HEC-RAS study LFRFLIKANA.prj: LFRFLIKANA

--- LFRFLIKANA.g01 (geometry) --- (continued)

Type RM Length L Ch R = 1 ,15428   ,106.6,113.9,120.9
XS GIS Cut Line= 4
2159040.90733428626712.6243392212159066.60259816626731.203991562
2159131.43372547 626769.944543252159141.71183102626786.152325079
#Sta/Elev= 30
       0 1685.43       4 1685.24       9 1685.21    17.1 1684.21    21.4 1683.95
    23.8 1684.04    31.4 1684.83    33.5 1684.81    40.1 1683.66    52.2    1682
      59 1680.25    60.5 1679.66    61.5 1679.34    63.5  1679.1    66.2    1679
    75.5 1679.75    80.1 1679.89    84.8 1679.63    89.5 1679.71    92.6 1680.55
    94.1 1681.09    98.8 1684.15   103.4 1688.17   107.2 1691.86   108.6 1692.93
   111.1  1694.6   115.9 1698.25   120.5 1700.19   123.6 1701.19   126.4 1701.63
#Mann= 3 ,-1,0
       0      .1       0    60.5    .045       0    75.5      .1       0
#XS Ineff= 2 , 0
           34.86 1693.96
Permanent Ineff=
       F       F
Bank Sta=60.5,75.5
XS Rating Curve= 0 ,0
Exp/Cntr(USF)=0,0
Exp/Cntr=0.3,0.1

Type RM Length L Ch R = 1 ,15315   ,77,73.9,71.8
XS GIS Cut Line= 4
2158981.49843629626750.3742012532158987.46335984626767.726706139
2159031.92915361626855.0314963442159025.96423005626912.511668777
#Sta/Elev= 30
       0 1683.23     7.2  1682.9    15.7 1682.91    24.5 1680.95    28.9 1680.48
    37.9 1679.87    43.8 1678.55    46.9 1677.39    51.4 1676.21    55.9 1676.99
    60.4 1678.21    64.9 1678.38    69.4 1677.31    73.8 1676.36    78.3 1675.85
    82.8 1676.01    90.4 1677.27    96.3 1678.43   103.2 1679.36   105.3 1679.81
   118.1 1683.81   122.5 1685.37     128 1687.01   136.3 1689.77   139.9 1690.85
   143.6 1691.74   150.7  1692.9   158.7 1694.45   165.4 1695.08   174.1 1695.64
#Mann= 3 ,-1,0
       0      .1       0    69.4    .045       0    90.4      .1       0
Bank Sta=69.4,90.4
XS Rating Curve= 0 ,0
Exp/Cntr(USF)=0,0
Exp/Cntr=0.3,0.1

Type RM Length L Ch R = 1 ,15241   ,87.7,83.7,80.4
XS GIS Cut Line= 4
2158912.63068252626782.9101479132158919.13787185626808.396639464
2158977.16031006626887.5674430042159008.06945939626911.969402999
#Sta/Elev= 30
       0 1682.58     6.5 1681.67    18.9 1680.68    30.5 1679.25    33.3 1678.68
    37.2 1677.52    44.8 1675.83    47.1 1675.17    50.5 1673.91    53.4 1673.08
    56.2 1672.58    59.1 1672.31      62    1672    66.9 1671.76    71.9 1671.72
    76.9 1671.86    80.8 1672.24    87.7 1672.78    91.7 1673.37    96.7  1675.2
   101.7 1676.74   106.6 1677.15   111.6 1677.23   116.5 1677.97   122.8    1680
   133.5 1684.41   146.4  1690.8   153.4 1693.95   159.3 1696.09   163.8 1697.11
#Mann= 3 ,-1,0
       0      .1       0    59.1    .045       0    80.8      .1       0
Bank Sta=59.1,80.8
XS Rating Curve= 0 ,0
Exp/Cntr(USF)=0,0
Exp/Cntr=0.3,0.1

Type RM Length L Ch R = 1 ,15157   ,77.6,81,79
XS GIS Cut Line= 4
2158851.89691542 626874.553064342158925.10279541626936.371362994
2158956.55421051626933.6600341062158989.63242295626942.878552327
#Sta/Elev= 30
       0 1685.52     2.1 1684.77     5.6 1683.13    10.6 1679.85    16.1 1675.59
    19.1 1674.16    21.3 1673.45    27.6 1672.37    36.1 1669.45    41.3 1669.18
    52.7 1668.47      58 1668.51    67.3  1669.3    70.2 1669.93      73 1670.95
    78.9 1673.52    84.1 1674.75    87.2 1675.14    98.9  1675.9   106.9 1676.87
     115 1678.18     127 1679.07   131.1 1680.35   135.3 1683.61   139.4 1685.96
   143.6 1687.44   149.4 1690.61   155.9 1693.89   160.2 1695.59   161.7 1695.94
#Mann= 3 ,-1,0
       0      .1       0    41.3    .045       0    67.3      .1       0
Bank Sta=41.3,67.3
XS Rating Curve= 0 ,0
Exp/Cntr(USF)=0,0
Exp/Cntr=0.3,0.1

Type RM Length L Ch R = 1 ,15076   ,101.4,105.9,107.7
XS GIS Cut Line= 4
2158817.57901903 626944.517331852158870.46666896626992.718734309
2158928.71003026627016.8194355392159043.27539141627022.750885897
#Sta/Elev= 30
       0 1680.89     5.1 1675.44       8 1673.21    22.1 1667.25    24.7 1666.48
    30.6 1665.69      36 1665.59    41.9 1665.95    46.41667.309    54.4 1671.24
    60.4 1672.63    71.6 1672.78    86.4 1673.77   103.8 1672.32   112.4 1672.18
   116.7 1672.52     121 1673.85   125.4 1675.87   142.1 1684.91   154.1 1692.19
   162.1 1694.81   171.7 1696.08   182.1 1698.18   194.1 1699.01   202.1 1700.17
     222 1700.66   226.2 1700.56   241.1 1698.74   246.2 1698.78   249.3  1699.3
#Mann= 3 ,-1,0
       0      .1       0    22.1    .045       0    46.4      .1       0
#XS Ineff= 2 , 0
                           63.66          1684.5
Permanent Ineff=
       F       F
Bank Sta=22.1,46.4
XS Rating Curve= 0 ,0
Exp/Cntr(USF)=0,0
Exp/Cntr=0.3,0.1

Type RM Length L Ch R = 1 ,14970   ,125.7,147.8,159.6
XS GIS Cut Line= 3
2158754.74258317627013.7327358422158848.11902592627136.006323745
 2158868.3511396627196.504317083
#Sta/Elev= 30
       0 1678.08     4.3 1677.17     9.2  1674.7    14.4 1669.83    15.5 1669.26
    24.5 1667.33    34.5 1663.35    37.7 1662.71    49.6 1661.23    54.7 1661.32
    61.81662.728    74.8 1664.37    81.4 1664.36    94.6 1663.06     105 1662.79
   117.6 1663.67   127.6 1663.06   134.2 1663.28   140.5 1664.63   147.4 1668.79
   150.3 1670.11     158 1674.43   173.8 1684.26   186.4 1692.25     193 1697.37
   197.3 1699.46   202.2 1701.26   209.9 1703.26   214.1 1704.77   217.6 1705.49
#Mann= 4 ,-1,0
       0      .1       0    37.7    .045       0    61.8      .1       0
  246.71     .08       0
Bank Sta=37.7,61.8
XS Rating Curve= 0 ,0
Exp/Cntr(USF)=0,0
Exp/Cntr=0.3,0.1

Type RM Length L Ch R = 1 ,14822   ,107.1,115.2,117.6
XS GIS Cut Line= 4
2158703.52859305626998.6697975732158705.33614565627093.867567431
2158701.72104046627202.3207229652158712.56635601627260.764923448
#Sta/Elev= 30
       0 1678.89     6.5 1676.77    22.5 1666.19    26.5 1664.56    30.5 1664.13
    50.5 1664.25    54.5 1664.73    62.5 1667.08    65.9 1667.15    74.5 1665.09
    77.7 1664.94    90.5 1666.36   110.5 1665.85   122.3 1664.67   130.5 1663.16
   134.5 1663.11   138.6  1661.4     143 1658.49   146.6 1657.67   158.6 1657.43
   174.6 1658.56   186.6 1661.09   198.6 1664.97   206.6 1668.47   214.8 1674.28
   218.8 1678.44     227 1688.59   239.2 1700.03   251.4 1706.87   263.2 1710.14
#Mann= 4 ,-1,0
       0      .1       0     143    .045       0   174.6      .1       0
  233.73     .08       0
Bank Sta=143,174.6
XS Rating Curve= 0 ,0
Exp/Cntr(USF)=0,0
Exp/Cntr=0.3,0.1

Type RM Length L Ch R = 1 ,14707   ,117.3,109.8,106.4
XS GIS Cut Line= 3
2158649.30201529626981.7993067122158627.00886665627023.975533864
2158574.58984147627202.320722965
#Sta/Elev= 30
       0 1674.71    15.2 1665.27    18.1 1663.77    21.1 1663.03    38.9  1662.8
      49 1663.14    53.1 1662.77    61.5 1661.35    71.9 1660.71    82.3 1659.13
    86.4 1658.81    90.7 1658.83      99 1659.49   111.5 1658.31     124 1658.36
   136.5 1654.55   140.7 1653.06   144.9 1652.58   161.5 1653.28   169.9 1654.27
   173.4 1654.38   186.3 1655.56   194.9 1655.11   199.1 1655.69   203.2 1657.96
   207.4 1661.43   211.6 1664.45   215.7 1666.32   219.9 1666.86   233.6 1666.38
#Mann= 3 ,-1,0
       0      .1       0   136.5    .045       0   173.4      .1       0
Bank Sta=136.5,173.4
XS Rating Curve= 0 ,0
Exp/Cntr(USF)=0,0
Exp/Cntr=0.3,0.1

Type RM Length L Ch R = 1 ,14597   ,70.4,64,58.1
XS GIS Cut Line= 4
2158497.44037488 626973.221931192158502.79608626627012.720302651
2158504.09529038627139.6588997682158491.44242223627189.065337289
#Sta/Elev= 30
       0 1688.12     9.5 1680.66    24.2 1671.57    36.3 1661.74    40.3 1659.21
    52.3  1655.2    64.3 1653.96    72.3 1653.94    79.3 1651.25    84.3 1650.32
   100.3  1649.7   104.3  1649.7   111.7 1651.17   120.3    1653   124.3 1652.55
   128.3 1651.18   132.3 1650.47   140.3 1650.17   144.3 1650.63   152.3 1653.87
   156.3  1654.2   160.3 1655.24   168.4 1660.31   172.5 1662.02   180.8 1663.57
     189 1666.64   193.1 1666.88   200.9 1666.01   209.7 1667.24   217.8 1666.38
#Mann= 3 ,-1,0
       0      .1       0    79.3    .045       0   111.7      .1       0
Bank Sta=79.3,111.7
XS Rating Curve= 0 ,0
Exp/Cntr(USF)=0,0
Exp/Cntr=0.3,0.1

Type RM Length L Ch R = 1 ,14533   ,92,85.3,76.7
XS GIS Cut Line= 3
2158421.55038866 627020.36042868 2158459.5089931627142.068969891
2158478.18703655627193.885477535
#Sta/Elev= 30
       0 1683.25       5 1679.11     9.2  1675.3    13.4 1671.22    17.6 1667.38
    30.2 1656.61    31.5 1655.68    34.4 1653.78    38.6 1652.16    44.3 1650.57
    50.7 1649.14    55.3 1648.57    63.7 1647.95    67.9 1647.96    72.1  1648.2
    88.6 1649.38    97.2 1650.91   105.6 1653.69   109.8 1654.44     114 1654.76
   118.2 1655.61   126.6 1660.79   127.3 1660.98   130.8 1661.48   139.3 1661.18
   147.8 1661.69   160.6 1663.31   164.8 1663.97   173.3 1665.61   182.6 1666.41
#Mann= 3 ,-1,0
       0      .1       0    50.7    .045       0    88.6      .1       0
Bank Sta=50.7,88.6
XS Rating Curve= 0 ,0
Exp/Cntr(USF)=0,0
Exp/Cntr=0.3,0.1

Type RM Length L Ch R = 1 ,14448   ,85.9,83.8,84.2
XS GIS Cut Line= 3
2158346.08418311 627092.746862332158390.54997688627153.480629429
2158434.47350487627208.249472974
#Sta/Elev= 30
       0 1669.84     5.5 1663.65    10.5 1657.02    15.4 1650.75    16.1 1650.15
      19 1648.56    20.4 1647.99    23.9 1647.54    36.1 1647.09      39 1647.06
    50.1  1647.3    55.1 1648.15    56.2 1648.63      60 1650.64    61.9 1651.29
      65 1652.01    74.9 1651.76    85.1 1652.73    90.4 1652.93      99 1652.96
   103.4 1653.24   104.7 1653.46   107.5 1654.34     116 1657.92   118.9 1658.62
     121 1659.02   130.3 1660.08     136  1660.9   141.7 1662.01   145.5 1662.93
#Mann= 3 ,-1,0
       0      .1       0      19    .045       0    56.2      .1       0
Bank Sta=19,56.2
XS Rating Curve= 0 ,0
Exp/Cntr(USF)=0,0
Exp/Cntr=0.3,0.1

Type RM Length L Ch R = 1 ,14364   ,68,79.2,95.9
XS GIS Cut Line= 3
 2158278.3009609627142.6353138762158357.47176444627246.208077411
2158378.07786399627279.828555627
#Sta/Elev= 30
       0 1660.48       6 1655.28    11.7 1651.05    13.3 1650.16    18.3 1648.31
    28.4 1646.65    34.5 1645.08    37.4 1644.51    43.5 1643.85    55.8  1643.6
    63.1 1643.93    68.7 1644.47    71.6 1645.01    75.5 1645.39    78.7 1645.33
    88.8 1644.69    93.8 1644.91    97.3 1645.59   103.9 1647.46     114 1651.75
     124 1656.39   128.7 1658.17   138.5 1660.42   143.2 1661.84   147.9 1662.78
   151.9 1663.26   154.9 1663.96   157.8 1664.84   166.7 1668.57   169.8 1669.69
#Mann= 3 ,-1,0
       0      .1       0    37.4    .045       0    68.7      .1       0
Bank Sta=37.4,68.7
XS Rating Curve= 0 ,0
Exp/Cntr(USF)=0,0
Exp/Cntr=0.3,0.1

Type RM Length L Ch R = 1 ,14285   ,93.5,98.8,107.9
XS GIS Cut Line= 3
 2158237.0887618627173.0021974262158250.64540624627277.659492516
2158243.59595113627323.752083618
#Sta/Elev= 30
       0 1649.55     4.2 1648.15     6.5    1648     8.2 1647.94    12.3 1648.53
    16.3 1648.73    20.8 1647.58      24 1646.61    27.9 1645.37    32.4 1643.67
    36.5 1642.45    44.5 1641.73    48.6 1641.63    56.6  1641.7    68.7 1641.23
    76.8 1641.91    81.5 1642.18    84.9 1642.77    88.9 1644.64    92.9 1646.99
      97 1648.98     101 1651.18     105 1654.33   113.1 1661.67   117.2 1664.81
   121.2 1667.14   125.3 1668.66   129.3 1669.75   138.9 1671.67   152.2  1675.1
#Mann= 4 ,-1,0
       0      .1       0    36.5    .045       0    81.5      .1       0
  152.16     .08       0
Bank Sta=36.5,81.5
XS Rating Curve= 0 ,0
Exp/Cntr(USF)=0,0
Exp/Cntr=0.3,0.1

Type RM Length L Ch R = 1 ,14186   ,78.1,79.1,81.1
XS GIS Cut Line= 3
2158154.98475443627156.392994326 2158137.9863491627270.638090632
2158137.19572559627286.845872461
#Sta/Elev= 30
       0 1647.25     4.8 1646.61     8.9  1645.7    12.9 1644.61    25.1  1642.8
    29.1 1642.02    33.1 1640.97    38.4  1639.8    45.3 1637.86    49.3  1637.4
    52.4 1637.36    57.4 1637.22    61.5 1636.98    65.5 1637.18    69.5 1637.12
    73.6 1636.94    80.6 1637.12    84.1 1637.39    93.8 1637.93    97.9 1638.39
   101.9 1640.39   105.3 1643.36   106.9 1644.99     110 1648.53     114 1652.83
     118 1656.43   122.1 1659.93   126.1 1663.13   130.1 1665.48   131.7 1665.98
#Mann= 3 ,-1,0
       0      .1       0    52.4    .045       0    84.1      .1       0
Bank Sta=52.4,84.1
XS Rating Curve= 0 ,0
Exp/Cntr(USF)=0,0
Exp/Cntr=0.3,0.1

Type RM Length L Ch R = 1 ,14107   ,82.5,81.7,78.8
XS GIS Cut Line= 3
2158080.64630885627145.0397096322158059.22346331627247.467689859
2158053.19828801 627267.55160755
#Sta/Elev= 30
       0 1659.82     3.9 1656.64     8.3 1652.71    12.4  1649.7    16.5 1647.04
    17.4 1646.34    20.6  1644.2    24.7 1641.02    28.7 1639.53    32.8 1638.93
    36.9  1637.7      41 1636.23    45.1 1634.93    53.3 1633.19    57.4 1632.33
    61.4 1631.97    65.5 1632.31    69.3 1633.17    73.7 1634.32    77.8 1635.21
    81.9 1635.11      86 1635.76    88.4 1637.15    91.8 1639.41    98.2 1644.32
   105.3 1648.87   114.9  1655.4     119 1657.91   123.1 1659.34   125.6 1659.74
#Mann= 3 ,-1,0
       0      .1       0    53.3    .045       0    69.3      .1       0
Bank Sta=53.3,69.3
XS Rating Curve= 0 ,0
Exp/Cntr(USF)=0,0
Exp/Cntr=0.3,0.1

Type RM Length L Ch R = 1 ,14026   ,103.3,103.3,102.5
XS GIS Cut Line= 3
2158000.98010201627102.1940185562157984.24350393627241.442514551
2157984.24350393627250.815009474
#Sta/Elev= 30
       0  1654.9       3 1652.61       7 1649.82    15.1 1644.82    19.1 1642.68
    23.2 1641.04    27.2 1639.74    31.2 1638.74    39.3 1636.04    43.3 1635.44
    51.4 1635.52    55.4 1634.78    59.4 1633.46    64.5 1632.54    66.6 1632.34
    71.5  1631.4    75.5 1630.96    87.6 1631.26   103.7 1631.31   107.8 1631.66
   111.3 1632.52   111.8 1632.63   115.8 1634.37   119.8 1637.14   123.9 1640.73
   131.9 1648.33     136 1651.71     140 1654.25     144 1655.66   149.6  1657.4
#Mann= 3 ,-1,0
       0      .1       0    66.6    .045       0   111.3      .1       0
Bank Sta=66.6,111.3
XS Rating Curve= 0 ,0
Exp/Cntr(USF)=0,0
Exp/Cntr=0.3,0.1

Type RM Length L Ch R = 1 ,13922   ,69.8,69.5,68.7
XS GIS Cut Line= 3
2157892.89979655627118.4803667892157888.01940456627200.470952373
2157887.53136536627236.585853166
#Sta/Elev= 22
       0 1646.44     2.7 1644.36    10.7 1636.91    14.7 1634.06    22.7 1632.41
    26.7 1631.37    34.8 1629.54    46.8 1627.36    50.8  1626.9    54.8 1626.73
    58.8 1626.43    62.8 1626.33    66.8 1627.29    70.8 1629.61    78.8 1633.19
    82.8 1635.63    91.1 1641.34    94.8 1643.71   102.8 1648.62   110.3 1651.69
   114.8 1653.77   118.3 1654.59
#Mann= 3 ,-1,0
       0      .1       0    46.8    .045       0    66.8      .1       0
Bank Sta=46.8,66.8
XS Rating Curve= 0 ,0
Exp/Cntr(USF)=0,0
Exp/Cntr=0.3,0.1

Type RM Length L Ch R = 1 ,13853   ,67.5,64.7,62.7
XS GIS Cut Line= 3
2157821.15803417627120.4325235882157820.18195577627206.815461971
2157824.57430857627236.585853166
#Sta/Elev= 30
       0 1641.08     1.7  1640.4     4.7 1638.94     8.7 1635.59    11.9 1633.76
    12.7 1633.23    16.7 1633.04    20.7 1633.08    24.7 1632.38    28.1 1630.59
    32.7 1627.81    36.7 1626.42    40.2 1625.85    44.3 1625.49    52.7 1625.17
      61 1625.48    68.8 1625.63    70.61625.886    72.8  1626.2    76.8 1627.58
    80.8 1629.95    84.7 1632.77    88.8 1635.54    92.8 1637.91    96.9 1640.53
   100.9 1643.89     105 1647.49     109 1650.16     113 1651.95   116.5 1652.29
#Mann= 3 ,-1,0
       0      .1       0    40.2    .045       0    70.6      .1       0
Bank Sta=40.2,70.6
XS Rating Curve= 0 ,0
Exp/Cntr(USF)=0,0
Exp/Cntr=0.3,0.1

Type RM Length L Ch R = 1 ,13788   ,70.9,72.4,73.8
XS GIS Cut Line= 3
2157753.17772178627137.991558094 2157759.3270157627221.446261278
2157765.47630962627249.118083912
#Sta/Elev= 29
       0 1634.68       2 1634.17     4.5  1633.7     7.2 1633.25    11.2  1632.8
    15.2 1631.48    19.2 1628.77    23.3 1626.24    27.3 1624.67    31.3 1624.04
    35.3 1623.62    40.31623.476    43.3 1623.43    47.3 1623.14    55.3 1623.55
    59.3 1623.47    63.4 1623.26    67.4 1623.25    71.4 1624.09    75.4 1625.72
    79.4 1628.42    84.2 1632.54    87.5 1635.56    91.6 1638.44    95.7 1640.92
    99.8    1643   103.9 1644.56     108 1645.63     112 1646.49
#Mann= 3 ,-1,0
       0      .1       0    40.3    .045       0    55.3      .1       0
Bank Sta=40.3,55.3
XS Rating Curve= 0 ,0
Exp/Cntr(USF)=0,0
Exp/Cntr=0.3,0.1

Type RM Length L Ch R = 1 ,13716   ,70.3,73.9,83.1
XS GIS Cut Line= 4
2157694.75942955627137.5523228142157685.53548867627163.467204329
2157682.46084171627226.7170846372157703.10489987627284.256906306
#Sta/Elev= 30
       0 1629.44       8 1628.54    12.3 1628.58    23.7  1627.9    29.2    1628
    33.2  1626.3    34.3 1625.51    37.2 1622.98    41.2 1621.81      451621.021
    49.2 1620.46    53.2 1620.54    57.3    1621    61.3 1620.96    65.3  1620.7
    69.3 1620.93    73.3 1621.59    81.3 1623.48    85.3  1625.3    89.3 1628.34
    93.4 1630.89   100.4 1633.81   106.2 1636.64   110.4 1637.93   118.9  1638.9
   123.2 1639.99   135.9 1644.94   140.2 1646.86   147.3 1650.38     152 1652.53
#Mann= 3 ,-1,0
       0      .1       0      45    .045       0    57.3      .1       0
Bank Sta=45,57.3
XS Rating Curve= 0 ,0
Exp/Cntr(USF)=0,0
Exp/Cntr=0.3,0.1

Type RM Length L Ch R = 1 ,13642   ,92.7,92.6,92
XS GIS Cut Line= 4
2157657.78786168627125.3129372172157619.32513083627157.205274651
2157599.44205231627226.4947906872157607.87729774627272.888640554
#Sta/Elev= 30
       0 1628.52     6.1 1628.36    12.3 1628.01    17.7  1627.3    31.1 1625.97
    43.7 1624.97    54.1 1624.33    58.3 1623.39    62.4 1621.98    70.7  1619.9
    74.9 1619.47    79.1 1619.68    91.3 1619.36    95.7 1619.38    99.9 1619.55
     104 1619.87   108.2 1621.02   112.4 1623.24   116.5 1625.79   126.1 1632.35
   128.8 1633.95   132.9 1635.92     137 1637.13     141 1638.06   145.1  1639.4
   149.3 1640.53   153.2  1641.2   157.3 1642.12   165.4  1643.7   169.2 1644.25
#Mann= 3 ,-1,0
       0      .1       0    70.7    .045       0     104      .1       0
Bank Sta=70.7,104
XS Rating Curve= 0 ,0
Exp/Cntr(USF)=0,0
Exp/Cntr=0.3,0.1

Type RM Length L Ch R = 1 ,13549   ,70.9,68.5,66.9
XS GIS Cut Line= 5
2157551.48027107627048.989993037 2157531.0366276 627094.01654106
 2157532.5626064627116.8366000912157515.08959801 627213.23940501
2157513.88456295627265.055912655
#Sta/Elev= 30
       0 1645.34       8 1643.94    13.4 1642.68    22.2 1639.96    32.9 1635.06
    39.7 1633.18    44.1 1630.82    48.5 1628.01    51.6 1627.02    56.6 1626.05
    68.7  1622.9    72.7 1622.35    74.5 1621.84    76.7 1621.16    88.9 1616.23
    93.6 1615.57   101.1 1615.47   113.3 1614.97   121.5 1615.44   137.7 1617.69
   141.8 1617.91   145.8 1617.65   149.9 1618.01     159 1621.49   166.2 1625.56
   169.3 1626.41   178.2 1627.47   182.2 1628.72   198.2 1635.55   222.1 1647.74
#Mann= 3 ,-1,0
       0      .1       0   101.1    .045       0   121.5      .1       0
Bank Sta=101.1,121.5
XS Rating Curve= 0 ,0
Exp/Cntr(USF)=0,0
Exp/Cntr=0.3,0.1

Type RM Length L Ch R = 1 ,13481   ,70.3,66.1,65.4
XS GIS Cut Line= 3
2157464.47812542627090.325828738 2157454.2353274627184.921081065
2157462.67057283627274.093675616
#Sta/Elev= 30
       0  1626.4     2.9 1624.25    10.9 1621.92    14.9 1619.92      19 1617.24
      23 1615.39      27 1614.22      31 1613.52    39.1 1613.19    59.2 1613.21
    65.81613.539    75.3 1614.34    79.3 1615.57    83.3 1617.59    87.4 1619.25
    91.4  1620.4    95.4 1620.98    99.4 1621.31   103.4 1621.28   115.7  1620.2
   127.6 1619.74   131.6  1619.8   135.6 1620.23   139.6 1621.23   143.6  1622.4
   147.6 1623.93   155.7 1628.19   170.6 1637.42   179.8 1643.77   184.7 1646.86
#Mann= 3 ,-1,0
       0      .1       0      31    .045       0    65.8      .1       0
Bank Sta=31,65.8
XS Rating Curve= 0 ,0
Exp/Cntr(USF)=0,0
Exp/Cntr=0.3,0.1

Type RM Length L Ch R = 1 ,13415   ,87,91.3,79.3
XS GIS Cut Line= 4
 2157391.5735042627088.5182761462157392.77853927627101.773661822
2157395.18860939 627189.13870378 2157401.2137847 627277.10626327
#Sta/Elev= 30
       0 1626.11     4.7 1622.74    12.7 1620.04    16.7  1618.2    24.7 1613.06
    28.7 1611.71    32.7 1611.73    40.7  1612.5    44.7 1612.27    48.7 1611.51
    52.7 1610.43    56.7 1609.74    64.7 1609.36    80.7 1610.23    84.7 1610.73
    87.4 1611.41    93.9 1613.39   100.7 1616.14   105.4 1617.39   109.2  1617.8
   128.8 1618.33   136.8 1617.92   144.9 1618.66   148.9 1619.53   152.9 1620.99
     158 1623.25   164.9 1626.63   176.9 1634.48   181.5 1637.14   188.9 1642.16
#Mann= 3 ,-1,0
       0      .1       0    48.7    .045       0    87.4      .1       0
Bank Sta=48.7,87.4
XS Rating Curve= 0 ,0
Exp/Cntr(USF)=0,0
Exp/Cntr=0.3,0.1

Type RM Length L Ch R = 1 ,13323   ,47.9,47.7,49.2
XS GIS Cut Line= 3
2157302.40090965 627116.234082562157343.97461928627215.649475133
2157356.62748742627278.913815862
#Sta/Elev= 30
       0 1620.07       1 1619.66     5.4 1618.66     9.7 1616.77    18.4 1611.04
    22.7 1609.06    26.5 1607.99    31.4 1607.64    35.7 1609.13      40 1611.06
    44.4 1611.68    53.1 1611.83    57.4 1610.66    61.7 1609.03    66.1 1608.42
    72.4  1608.1    87.7 1608.07    92.1 1608.71    96.9 1610.32   100.7 1612.48
   105.1 1614.49   112.6 1615.89   125.6 1617.12   133.8  1619.1   137.9 1620.42
     142 1622.27   150.1 1627.72   158.3 1631.53   170.4 1639.52   172.3  1640.5
#Mann= 3 ,-1,0
       0      .1       0    18.4    .045       0      40      .1       0
Bank Sta=18.4,40
XS Rating Curve= 0 ,0
Exp/Cntr(USF)=0,0
Exp/Cntr=0.3,0.1

Type RM Length L Ch R = 1 ,13276   ,67.7,65.7,61.5
XS GIS Cut Line= 3
2157265.86026648627145.8468814512157297.48520664627226.885790595
2157316.06485898627276.299759585
#Sta/Elev= 30
       0 1612.91     3.6 1611.24     7.9 1609.68    16.5 1607.33    19.2 1606.87
    20.8 1606.65    29.3 1606.12    33.6  1606.2    41.4 1606.98    44.5 1606.98
    50.8 1606.65    55.1 1606.61    61.4 1607.15    63.7 1607.59      68 1608.76
    72.3 1610.53    76.6 1611.98    80.9 1612.74    85.2 1613.13    89.4 1614.04
    93.7 1615.24      98 1616.89   102.3 1618.99     106    1621   110.8 1623.48
   115.1 1625.32   119.4 1627.57   123.6 1629.52   131.2 1632.78   139.8 1636.83
#Mann= 3 ,-1,0
       0      .1       0    19.2    .045       0    41.4      .1       0
Bank Sta=19.2,41.4
XS Rating Curve= 0 ,0
Exp/Cntr(USF)=0,0
Exp/Cntr=0.3,0.1

Type RM Length L Ch R = 1 ,13210   ,64.6,84.8,84.1
XS GIS Cut Line= 4
2157218.06279178627155.0713645932157205.77288019 627182.61087438
2157242.53687312627236.373272641 2157279.6961778627262.463848268
#Sta/Elev= 30
       0 1613.32       3 1612.73    11.1 1611.51    15.4 1610.59    19.8  1609.1
    24.2 1607.03    27.3 1605.98    33.3 1604.59    36.6 1603.45    39.5  1602.7
    45.2  1601.4    47.8 1600.79    52.7 1600.29    55.7 1600.54    59.6 1601.21
    62.3 1601.68    67.2 1602.96    71.1 1604.65    76.9 1607.56    81.7  1609.3
    86.6 1609.95    95.3 1610.35   102.2 1610.92   108.5 1611.89   114.3 1613.12
   121.7  1615.9   126.6 1616.95   131.5  1618.5   136.4 1620.49   140.7 1622.57
#Mann= 3 ,-1,0
       0      .1       0    45.2    .045       0    59.6      .1       0
Bank Sta=45.2,59.6
XS Rating Curve= 0 ,0
Exp/Cntr(USF)=0,0
Exp/Cntr=0.3,0.1

Type RM Length L Ch R = 1 ,13125   ,70.9,85.2,83.3
XS GIS Cut Line= 2
 2157162.0636562627130.3102445722157127.31630435627281.563423228
#Sta/Elev= 30
       0 1610.74       7 1611.11    11.2  1610.5      14 1608.79    15.3 1607.84
    23.5 1601.09    27.3 1597.62    31.7 1594.22    35.8 1593.08    39.9 1593.33
      44 1593.22    48.1 1593.48    56.3 1595.11    60.71596.264    64.5 1597.41
    68.6 1597.03    72.7 1595.97    77.21595.533      85 1594.67    89.1 1594.48
    94.1 1594.48   101.4 1594.01   105.5 1594.05   117.9  1594.8   126.1 1596.35
   130.2 1597.62   138.4 1600.49   142.5 1602.17   150.8  1606.1   155.2 1607.82
#Mann= 1 ,-1,0
       0   -9999       0
Bank Sta=60.7,77.2
XS Rating Curve= 0 ,0
Exp/Cntr(USF)=0,0
Exp/Cntr=0.3,0.1

Type RM Length L Ch R = 1 ,13040   ,66.5,76.9,71.9
XS GIS Cut Line= 2
2157115.73385373627120.7717558272157006.04123317627263.167766364
#Sta/Elev= 30
       0 1605.65     8.5 1604.47    12.4 1603.47    15.7 1601.98    25.6 1595.48
    30.8 1593.15    38.6 1590.31    42.8 1589.16    45.2 1588.73    55.51587.693
    64.8 1585.95    71.2 1585.44    77.41585.574    82.7 1585.74    86.4  1586.3
    88.4 1586.88    91.2 1588.05    96.4 1590.86    97.6 1591.33   108.4 1594.27
   114.1 1596.04   121.7 1598.73   131.8 1602.98   136.9 1604.43   141.9 1605.13
     152 1605.61   156.6 1605.42   162.5 1604.57   168.3 1604.13   179.7 1604.01
#Mann= 1 ,-1,0
       0   -9999       0
Bank Sta=55.5,77.4
XS Rating Curve= 0 ,0
Exp/Cntr(USF)=0,0
Exp/Cntr=0.3,0.1

Type RM Length L Ch R = 1 ,12963   ,70.2,70.9,70.8
XS GIS Cut Line= 4
2157084.69663629627081.991792988 2157063.7109507627093.216694586
2156995.87350191627151.7813985752156973.91173791627246.461003357
#Sta/Elev= 30
       0 1612.62     9.7 1608.91    14.2 1606.17    29.9 1592.85    34.8 1587.48
    37.6 1585.58      39 1584.95    43.3 1584.45    57.5 1583.58    70.7 1584.18
    74.5 1583.04    80.2 1582.02    81.3 1582.04    85.8 1584.24    88.7 1585.57
    97.2 1588.44   102.5 1589.53   107.7 1589.72     119 1588.38   127.2 1588.26
   131.3 1588.52   143.6 1590.19   155.9 1592.21     161  1593.3   164.1 1594.35
   176.4 1599.57   184.7 1601.78   188.8  1602.3     197 1602.43   210.6 1601.66
#Mann= 3 ,-1,0
       0      .1       0    43.3    .045       0    85.8      .1       0
Bank Sta=43.3,85.8
XS Rating Curve= 0 ,0
Exp/Cntr(USF)=0,0
Exp/Cntr=0.3,0.1

Type RM Length L Ch R = 1 ,12892   ,77.5,66.1,51.4
XS GIS Cut Line= 3
2157054.57424081627010.6805587922156934.25624957627110.775314949
2156952.91537204627235.804210911
#Sta/Elev= 30
       0 1612.21     6.3 1606.68    16.4 1599.45    49.9 1579.94    54.6 1579.03
    73.5 1578.44    81.2 1577.04    91.5 1576.35    97.2 1576.54   102.51577.849
   110.2 1580.53   122.8  1583.5   141.5 1591.52   147.8 1592.87   167.4 1591.59
   177.9 1590.25   187.3 1587.79   195.3 1583.28     199 1582.19   207.5 1582.19
   211.5 1583.77   219.6 1588.37   231.7    1592   243.9 1597.58   247.9 1598.78
     252 1599.74   264.1 1600.75   272.2 1602.49   276.2 1602.65   282.9 1601.69
#Mann= 3 ,-1,0
       0      .1       0    80.3    .045       0   108.8      .1       0
#XS Ineff= 1 ,-1
  139.44   278.2 1601.23
Permanent Ineff=
       F
Bank Sta=73.5,102.5
XS Rating Curve= 0 ,0
Exp/Cntr(USF)=0,0
Exp/Cntr=0.3,0.1

Type RM Length L Ch R = 1 ,12826   ,199,182.6,155.6
XS GIS Cut Line= 5
2156966.11140514626919.9987936682156954.73051845 626955.48038159
2156921.25732229627110.1265478152156895.81769322627169.039373044
2156895.14822929627221.257559042
#Sta/Elev= 30
       0 1630.36      39  1595.1    44.2 1591.07    59.5 1580.61    67.6 1576.72
    71.7 1576.01    79.9 1575.39    87.9 1576.21    91.3 1575.31    96.3 1574.44
   104.8 1574.14   120.9 1575.07     129 1575.74   137.2 1579.01   141.3  1580.1
   153.6 1581.06   158.6    1582     162 1583.18   175.4  1591.1   182.2 1593.31
   188.9 1592.95   229.1  1586.6   246.7 1582.67   251.1 1582.32   263.8 1583.77
   283.8 1584.26   291.8 1587.26   303.8 1596.17   307.8 1598.37   311.9 1599.17
#Mann= 3 ,-1,0
       0      .1       0    91.3    .045       0   120.9      .1       0
Bank Sta=91.3,120.9
XS Rating Curve= 0 ,0
Exp/Cntr(USF)=0,0
Exp/Cntr=0.3,0.1

Type RM Length L Ch R = 1 ,12643   ,120.9,122.5,115.3
XS GIS Cut Line= 4
2156729.21749528626973.8282639942156800.89699752627046.016558817
2156841.73429683627116.9797346612156853.11518352627219.407714888
#Sta/Elev= 30
       0 1585.22    10.1 1576.16    12.9  1574.3    15.6 1573.04    18.6 1572.81
    29.9 1573.55    41.2 1572.17    52.5 1570.97    63.9 1570.73    72.4 1571.44
    75.2 1572.34    80.8 1574.15    89.3 1575.44   103.5 1575.57   128.5 1576.86
   151.5 1576.52   156.2 1577.22   166.6 1579.76   183.8 1582.33   195.9 1582.05
   211.4  1580.2   236.1 1579.17   240.2 1579.78   248.2 1582.13   256.2 1582.68
   260.3 1583.45   264.3 1585.13   272.3 1590.35   276.1  1592.1   286.7 1595.38
#Mann= 3 ,-1,0
       0      .1       0    41.2    .045       0    75.2      .1       0
Bank Sta=41.2,75.2
XS Rating Curve= 0 ,0
Exp/Cntr(USF)=0,0
Exp/Cntr=0.3,0.1

Type RM Length L Ch R = 1 ,12521   ,101.3,94.5,78.1
XS GIS Cut Line= 4
2156661.24001278627057.5125714792156743.32310014627130.369013122
2156772.77951275627173.2147041972156802.23592537627235.474849041
#Sta/Elev= 30
       0 1585.79     5.5 1581.41    14.6 1574.92    18.8 1573.15    38.7  1570.4
    46.7 1570.48    52.1 1569.99      67 1567.54    75.5 1566.59    89.9 1566.44
    95.3 1566.67    98.2  1567.4     108 1572.07   111.3 1572.87   113.2 1572.84
     118 1571.54   123.9    1569   127.7 1568.16   132.6 1568.99   138.3 1571.14
     152 1574.68   155.5 1574.94   161.7 1574.79   173.3 1575.96   200.3 1584.08
   201.5 1584.57   210.4 1590.05   214.8  1591.4   219.2  1591.9   230.6 1591.17
#Mann= 3 ,-1,0
       0      .1       0      67    .045       0    98.2      .1       0
Bank Sta=67,98.2
XS Rating Curve= 0 ,0
Exp/Cntr(USF)=0,0
Exp/Cntr=0.3,0.1

Type RM Length L Ch R = 1 ,12427   ,84.5,91.5,95.8
XS GIS Cut Line= 3
2156616.12495476627177.2314877352156713.86668752627192.629157966
2156761.39862606627235.474849041
#Sta/Elev= 30
       0 1576.37     4.1 1575.01     8.1 1574.12    16.2 1574.31    20.3 1573.86
    24.2 1573.17      35 1569.88      42 1567.56    45.5 1566.36    48.6 1565.48
    52.7  1565.2    60.8 1566.25    66.5 1566.66    73.5 1567.46      77 1568.28
    85.1 1570.68    89.1 1571.59    99.8 1572.93   103.8 1573.93   105.7 1574.62
   109.5  1576.4   112.3 1578.03   115.1 1580.05   117.7 1582.11   123.6 1585.87
     129 1587.12   132.1  1587.3   147.6  1589.1   155.9 1589.54   162.9 1589.68
#Mann= 3 ,-1,0
       0      .1       0      42    .045       0    73.5      .1       0
Bank Sta=42,73.5
XS Rating Curve= 0 ,0
Exp/Cntr(USF)=0,0
Exp/Cntr=0.3,0.1

Type RM Length L Ch R = 1 ,12335   ,106.9,114,121.4
XS GIS Cut Line= 3
2156593.83625312627248.7055382022156666.17830372627280.330478356
2156702.15167315627302.863248216
#Sta/Elev= 30
       0 1571.17     2.6 1570.24     8.2 1567.83    15.6 1565.01      20 1563.17
    24.4 1560.72    26.4 1559.84    28.7 1558.82    31.1 1558.37    33.1 1558.15
    37.5  1558.4    41.8 1558.85    46.2 1558.73    50.7 1558.83    53.8 1559.12
    56.8  1559.6    59.3 1560.09    63.7 1561.27      68 1563.33      69 1563.94
    72.4 1566.34    80.6 1571.09    90.7 1578.16    95.5  1581.1   103.2 1584.23
   107.1 1585.64   110.7 1586.61   114.3 1588.15   118.7 1589.61   121.4 1590.14
#Mann= 3 ,-1,0
       0      .1       0    26.4    .045       0    56.8      .1       0
Bank Sta=26.4,56.8
XS Rating Curve= 0 ,0
Exp/Cntr(USF)=0,0
Exp/Cntr=0.3,0.1

Type RM Length L Ch R = 1 ,12221   ,103.7,115.4,130.5
XS GIS Cut Line= 4
2156555.61276464  627332.67823272156569.44867596627345.723520513
2156612.93296867627400.6718540312156641.79072656627442.574899735
#Sta/Elev= 30
       0 1566.91      .8 1566.91     3.6 1566.42     6.6  1565.7    12.4 1563.11
    17.3 1562.13    23.4 1561.44    28.5 1560.29    29.9 1559.87    37.7 1556.53
    40.5 1555.97    43.3 1555.66    48.9 1555.56      54 1555.77    57.6 1556.34
    68.5 1557.48    71.8 1557.65    74.4 1558.14      75 1558.43    77.5 1560.23
    80.4 1562.61    89.7 1571.07    94.6 1574.75   101.9 1581.21   109.1 1587.06
     114  1591.4     116 1593.29   118.8 1596.27   123.7 1600.84     140 1614.26
#Mann= 3 ,-1,0
       0      .1       0    37.7    .045       0    57.6      .1       0
Bank Sta=37.7,57.6
XS Rating Curve= 0 ,0
Exp/Cntr(USF)=0,0
Exp/Cntr=0.3,0.1

Type RM Length L Ch R = 1 ,12106   ,112.7,117.7,129.3
XS GIS Cut Line= 4
 2156484.4566493627357.1875613192156484.06133755627380.510954683
2156477.34103776627448.8998877662156478.13166127627492.779492229
#Sta/Elev= 30
       0 1561.17       4 1561.44      12 1561.56      16 1561.12    24.2 1558.35
      28 1557.27    31.2 1555.82    34.8 1553.64    36.1 1552.95    40.1 1551.49
    48.1  1549.9    52.1  1549.4    56.2  1549.3    60.4 1549.65    64.2 1550.36
    68.2 1550.88    72.2 1551.37    76.2 1553.41    77.7 1554.72    78.7 1555.76
    84.3 1560.77    88.3 1563.58    92.3 1567.24    96.3 1571.38   100.3 1574.82
   104.3 1577.83   108.3  1580.5   124.3 1592.07   132.3 1597.45   135.9 1599.38
#Mann= 3 ,-1,0
       0      .1       0    40.1    .045       0    68.2      .1       0
Bank Sta=40.1,68.2
XS Rating Curve= 0 ,0
Exp/Cntr(USF)=0,0
Exp/Cntr=0.3,0.1

Type RM Length L Ch R = 1 ,11988   ,77.5,76.3,72.7
XS GIS Cut Line= 4
2156418.30781614627332.9856973962156380.48965854627358.373496575
 2156351.2365889627401.8577892872156344.12097736627452.062381781
#Sta/Elev= 30
       0 1556.89    21.9 1556.06    26.7 1555.22    30.5 1554.24    33.4 1553.87
    36.3 1553.91    39.2 1553.68    43.4 1554.06    48.9    1554    56.4 1551.04
    59.3 1550.09    62.2 1549.21    65.1  1548.6      73 1547.58    77.9 1548.04
    81.9 1549.91    82.7 1550.23    87.5 1553.29    89.1 1553.76    93.9 1554.59
      98 1555.76   101.3 1557.03   113.4 1562.34   117.5 1564.33   121.5 1566.87
   125.6 1569.94   133.6 1577.15   137.7 1579.89   141.7 1581.47   148.7 1583.23
#Mann= 3 ,-1,0
       0      .1       0    59.3    .045       0    81.9      .1       0
Bank Sta=59.3,81.9
XS Rating Curve= 0 ,0
Exp/Cntr(USF)=0,0
Exp/Cntr=0.3,0.1

Type RM Length L Ch R = 1 ,11912   ,71.6,69,64.4
XS GIS Cut Line= 4
2156348.33550485 627276.634397962156315.14883926627315.189494753
2156283.42629127 627379.122629942156288.30668326627416.213609133
#Sta/Elev= 30
       0 1554.08     6.4 1553.45    11.3 1552.39    16.6 1550.79    20.4 1550.27
      26 1550.13    37.7 1550.34    53.1 1549.66    57.6 1549.03    60.5 1547.82
    65.81546.024      71 1544.99    75.4 1544.75    79.9  1544.7    84.3 1544.87
    88.8 1545.24      93 1546.12    97.7 1546.62    99.3 1547.15   102.2 1548.38
   111.1 1556.32   115.6 1558.81   117.2  1559.3   120.1 1560.11   122.2  1560.5
   136.4 1562.77   144.5  1564.3   148.5 1564.66   156.6 1565.82   159.7 1566.08
#Mann= 3 ,-1,0
       0      .1       0    65.8    .045       0      93      .1       0
Bank Sta=65.8,93
XS Rating Curve= 0 ,0
Exp/Cntr(USF)=0,0
Exp/Cntr=0.3,0.1

Type RM Length L Ch R = 1 ,11843   ,75.1,72.2,69.1
XS GIS Cut Line= 4
2156269.27315447627239.5434187672156262.92864487627256.136751564
2156228.27786168627353.2565523452156224.86158728627373.266159541
#Sta/Elev= 30
       0  1555.6       6 1553.81    10.3 1553.13    14.6 1551.92    23.1 1547.59
      27 1546.51    31.6 1545.79    40.1 1545.06    44.4 1544.54    48.9 1543.63
    52.8 1543.28    55.2 1543.23    61.3 1543.38    65.6 1542.96    73.9 1543.64
    78.3 1543.13    82.6    1543    86.8 1543.67    91.1 1545.66    95.3 1547.94
    99.6 1548.74   103.8 1549.03   108.4 1549.52   116.6 1551.16   120.9 1553.24
   124.9 1556.04   128.9 1558.56     133 1559.82     137 1559.81   141.2 1559.15
#Mann= 3 ,-1,0
       0      .1       0    48.9    .045       0    86.8      .1       0
Bank Sta=48.9,86.8
XS Rating Curve= 0 ,0
Exp/Cntr(USF)=0,0
Exp/Cntr=0.3,0.1

Type RM Length L Ch R = 1 ,11770   ,71.7,72.9,73.6
XS GIS Cut Line= 4
2156207.76512752627220.2806520082156188.73159872627238.338102404
2156170.18610912627318.3765311892156166.76983472627354.979471182
#Sta/Elev= 30
       0 1553.36    10.5  1551.8      16 1550.32    20.2 1548.95    26.2 1546.54
    33.3 1544.15    37.4 1542.59    41.5 1540.81    45.6 1539.66    49.7 1539.12
    57.9 1537.63      62  1537.1    66.1 1536.94    70.2 1537.54    74.3 1538.65
    78.4 1539.56    82.5 1540.78    86.6 1542.49    90.7 1543.87    94.8 1544.43
      99 1544.81   115.2 1545.47   119.2 1545.83   123.3 1546.87   127.5 1549.13
   131.3 1550.97   135.3 1552.57   139.3 1553.99   143.3 1555.01   145.2 1555.19
#Mann= 3 ,-1,0
       0      .1       0    41.5    .045       0    82.5      .1       0
Bank Sta=41.5,82.5
XS Rating Curve= 0 ,0
Exp/Cntr(USF)=0,0
Exp/Cntr=0.3,0.1

Type RM Length L Ch R = 1 ,11698   ,113.9,108.3,107.1
XS GIS Cut Line= 2
2156125.24644623627199.7676663062156089.64839802627331.503661354
#Sta/Elev= 30
       0 1555.79     8.5 1553.34      18 1550.99    22.2 1549.52    24.9 1548.04
    30.5 1544.65    37.2 1541.45    38.8 1540.77    42.9 1539.38    55.3 1536.39
    59.5 1536.49    67.8 1538.64    75.51540.353    77.1 1540.78      80 1541.83
    84.3 1542.88    90.1 1543.79    92.6 1543.94    93.4 1543.91    96.8 1543.29
   100.9 1541.58     105 1541.84   106.4 1542.13   109.2 1542.94   113.3 1543.84
   117.5 1546.17   121.6 1549.21   125.8 1550.51   132.5 1550.54   136.5  1550.7
#Mann= 3 ,-1,0
       0      .1       0    23.8    .045       0    62.5      .1       0
#XS Ineff= 1 ,-1
    70.2     125 1548.18
Permanent Ineff=
       F
Bank Sta=37.2,75.5
XS Rating Curve= 0 ,0
Exp/Cntr(USF)=0,0
Exp/Cntr=0.3,0.1

Type RM Length L Ch R = 1 ,11589   ,99.6,106.6,114.6
XS GIS Cut Line= 4
2156031.58297635627189.5341824132156007.66905555627212.960064009
2155994.98003636627281.2855519962156010.10925155627308.127707991
#Sta/Elev= 30
       0 1549.66     2.2 1548.02     4.8 1546.29     7.8 1543.62    10.6 1541.69
    13.5 1540.61    16.3  1539.9      22 1539.03    27.2 1538.79    32.8 1538.79
    37.8 1538.43    41.8 1537.28    45.9 1535.64      50 1534.87    53.8 1534.66
    58.11534.581    66.2 1534.31    70.3  1534.3    78.5 1534.66    82.5 1534.96
    86.6 1536.16    94.7 1540.88    98.8  1542.1   102.9 1542.37     112 1542.28
   116.6 1543.18   121.2 1544.91   125.8 1545.64   130.4 1545.51   133.8 1545.68
#Mann= 3 ,-1,0
       0      .1       0    58.1    .045       0    78.5      .1       0
Bank Sta=58.1,78.5
XS Rating Curve= 0 ,0
Exp/Cntr(USF)=0,0
Exp/Cntr=0.3,0.1

Type RM Length L Ch R = 1 ,11483   ,126.6,123.3,119
XS GIS Cut Line= 3
2155950.56846916627149.5149680212155904.69278437 627207.10359361
2155877.85062838627270.060650398
#Sta/Elev= 30
       0 1541.66     9.8 1535.61    14.9 1533.42    21.4 1531.89    23.1 1531.34
    29.5 1529.72    32.41529.456    40.5 1529.11    47.21529.376    55.8 1529.48
    60.9 1530.14    66.1 1532.11    69.8 1533.72    71.2 1534.12    72.6 1534.24
    75.9 1534.21    84.6 1531.44    88.9 1530.84    93.9 1531.25    97.6 1531.39
     100 1531.69     102  1532.1   109.1 1535.09   110.7 1535.58     115 1536.27
   119.4 1536.57   123.7 1536.66   128.1 1536.55   136.8 1536.62   142.1 1536.46
#Mann= 3 ,-1,0
       0      .1       0    32.4    .045       0    47.2      .1       0
Bank Sta=32.4,47.2
XS Rating Curve= 0 ,0
Exp/Cntr(USF)=0,0
Exp/Cntr=0.3,0.1

Type RM Length L Ch R = 1 ,11359   ,154.2,151.1,143.6
XS GIS Cut Line= 3
2155857.06005436627046.5912190112155836.50384326627086.913017707
 2155774.4398982627229.620560152
#Sta/Elev= 30
       0 1573.97    20.9 1558.31    25.4 1554.63    29.8 1550.68    34.3 1547.16
    43.3 1543.19    47.7 1539.28    56.5 1529.75    60.8  1525.7    65.2 1523.82
    69.5 1523.23    80.7 1522.96      87 1523.09    98.9 1523.87   104.4 1524.75
   108.8 1525.95   117.1 1529.33   121.9 1529.91   132.3 1530.01   135.4 1529.58
   139.3 1528.25   144.5 1526.91   148.1 1526.46   152.4 1526.66   161.1 1529.31
   171.9 1531.48   174.2 1531.72   178.6 1531.61   190.1 1531.96   200.9 1532.51
#Mann= 3 ,-1,0
       0      .1       0    65.2    .045       0    98.9      .1       0
#XS Ineff= 2 , 0
                          117.61          1549.7
Permanent Ineff=
       F       F
Bank Sta=65.2,98.9
XS Rating Curve= 0 ,0
Exp/Cntr(USF)=0,0
Exp/Cntr=0.3,0.1

Type RM Length L Ch R = 1 ,11208   ,140.7,132.4,121
XS GIS Cut Line= 4
2155692.70885337 627018.274310612155684.27360794627049.605222209
2155663.78801189627165.2885881132155648.12255609627226.142858719
#Sta/Elev= 30
       0 1563.68     7.2 1559.46    19.6 1550.67    23.7 1546.21    27.9 1541.24
    32.4 1536.54    44.2 1526.15    48.3 1522.76    51.5 1520.58    52.3 1520.05
    56.4    1519    60.4 1518.81      77 1519.03    80.8 1519.46    83.9 1520.73
    88.9 1523.15    92.9 1524.55      97 1525.72   101.1 1526.52   105.1 1526.86
   109.2 1526.96   117.3 1526.62   133.6 1526.41   141.7 1526.71   149.8 1527.49
   162.2  1528.2   174.6 1527.78     187 1527.83   199.4 1528.34   212.8 1528.16
#Mann= 3 ,-1,0
       0      .1       0    51.5    .045       0    83.9      .1       0
Bank Sta=51.5,83.9
XS Rating Curve= 0 ,0
Exp/Cntr(USF)=0,0
Exp/Cntr=0.3,0.1

Type RM Length L Ch R = 1 ,11076   ,120.5,113.8,100.4
XS GIS Cut Line= 4
2155538.25133291626989.1620377562155539.59026076627036.693976293
2155576.41077653627190.6706785962155599.17254991627243.558328518
#Sta/Elev= 30
       0 1530.52      16 1530.03      28  1529.2      36 1528.82      48 1529.04
    52.2 1528.94    56.3 1527.76    60.4  1524.6    64.5 1520.82    68.6 1518.83
      69 1518.75    72.7 1517.94    81.6 1517.82    89.2 1517.99   104.9    1518
   109.7 1518.58     118 1522.22   122.1 1522.72   128.1 1522.74   146.8 1521.95
   167.3 1521.66   179.7 1521.65   191.2 1522.92   204.3 1524.87     213 1525.86
   217.3 1526.01   230.4 1525.95   239.1 1526.54   250.2 1526.44   263.4 1526.77
#Mann= 3 ,-1,0
       0      .1       0      69    .045       0   109.7      .1       0
Bank Sta=69,109.7
XS Rating Curve= 0 ,0
Exp/Cntr(USF)=0,0
Exp/Cntr=0.3,0.1

Type RM Length L Ch R = 1 ,10962   ,102,105.6,97.9
XS GIS Cut Line= 3
 2155407.0129922627072.4401798392155537.18653279627231.623823766
2155573.63512416627289.644030431
#Sta/Elev= 30
       0  1541.3    15.6 1540.96    20.8 1540.06    24.1 1537.73    26.8 1535.39
    33.4 1528.18    37.1 1524.97    39.7 1522.98    46.8 1518.08    52.4 1516.04
    55.4  1515.5    58.2 1515.12      63 1514.97    78.1 1515.04      84 1515.52
    92.3 1518.34    96.6 1518.94   106.5 1519.31   166.3 1519.94   171.9 1520.47
   174.7 1520.98   181.8 1522.99     187 1523.98     204 1524.64   213.8 1525.25
   226.3    1525   240.5 1525.11   252.4 1525.63   264.2 1525.79   274.2 1526.29
#Mann= 3 ,-1,0
       0      .1       0    55.4    .045       0      84      .1       0
Bank Sta=55.4,84
XS Rating Curve= 0 ,0
Exp/Cntr(USF)=0,0
Exp/Cntr=0.3,0.1

Type RM Length L Ch R = 1 ,10856   ,140.4,136.4,137.4
XS GIS Cut Line= 2
2155363.68217706627179.8174989282155540.09312448627317.798209484
#Sta/Elev= 30
       0  1535.8     8.7 1534.88    10.8 1534.31    15.2 1533.77    20.9 1532.71
    21.7 1532.22      26 1528.55    35.5 1518.71    38.4 1516.51      391516.199
    41.3 1515.03    49.8 1514.05    66.6 1513.76    71.7 1513.99    83.4 1514.89
    92.5 1515.47   102.2 1516.41   112.6 1516.52   117.4 1517.69   125.6 1521.33
   129.5 1522.29   132.1 1522.46   146.6 1522.64     153 1523.28     158 1523.53
   164.5 1523.38   169.4 1523.47   195.1 1524.88     215  1525.5     224 1525.44
#Mann= 3 ,-1,0
       0      .1       0      32    .045       0    78.6      .1       0
Bank Sta=39,83.4
XS Rating Curve= 0 ,0
Exp/Cntr(USF)=0,0
Exp/Cntr=0.3,0.1

Type RM Length L Ch R = 1 ,10720   ,62.1,59.5,60.8
XS GIS Cut Line= 2
2155288.27350719627266.7362271672155430.03257023627416.703963493
#Sta/Elev= 30
       0 1525.63     7.3 1522.72    17.3 1520.26    19.9 1519.32    24.3 1517.03
    27.1  1515.8      30  1515.1    36.4 1514.74    58.2 1515.01    69.6  1515.4
    85.9 1513.89    93.3 1512.25    96.9 1511.39    98.8 1511.17   106.4 1511.03
   115.71511.112   118.9 1511.19   120.5  1511.4   123.3 1512.23   124.5 1512.81
   126.2 1513.94   131.8 1518.69   134.6 1520.19   137.5 1520.65   145.4 1521.06
     152 1521.75   157.5 1521.95   179.5 1521.92     196 1521.47   206.4 1521.84
#Mann= 3 ,-1,0
       0      .1       0    85.1    .045       0   108.2      .1       0
Bank Sta=93.3,115.7
XS Rating Curve= 0 ,0
Exp/Cntr(USF)=0,0
Exp/Cntr=0.3,0.1

Type RM Length L Ch R = 1 ,10661   ,101.7,102.4,95.8
XS GIS Cut Line= 5
2155246.16591344627313.0621115392155302.40088298627358.585658307
2155312.44284182627373.9833285372155360.64424428627411.473308228
2155396.79529613 627446.95489615
#Sta/Elev= 30
       0 1522.54      10 1519.91    12.9    1519    18.6 1515.96    21.4 1514.86
    23.2 1514.45    25.6 1514.28    33.5 1514.46    38.5 1514.27    44.2 1513.46
      54  1512.8    57.4 1512.11    64.3 1510.24    70.1 1509.51    75.4 1509.56
    88.21510.174   100.5 1510.53     109 1510.56   112.8 1510.98   115.5 1511.56
     122 1515.76     127 1517.86   128.5 1518.24   138.4 1519.76   149.8 1520.78
   152.7 1520.86   178.1 1520.08   182.8 1520.38   197.9 1522.47   202.5 1522.75
#Mann= 3 ,-1,0
       0      .1       0    64.3    .045       0    88.2      .1       0
Bank Sta=64.3,88.2
XS Rating Curve= 0 ,0
Exp/Cntr(USF)=0,0
Exp/Cntr=0.3,0.1

Type RM Length L Ch R = 1 ,10558   ,88.6,81.6,69.4
XS GIS Cut Line= 2
2155183.46246161627375.4432762212155286.19432878627468.129680307
#Sta/Elev= 30
       0 1522.46     2.6 1520.92     6.3 1519.01    13.1 1516.57    15.9 1515.36
    22.5 1511.68    24.4 1510.71    26.41509.929    27.9 1509.54    32.4 1509.23
    38.6 1509.28    49.4 1509.12    55.5  1509.2    59.41509.449    62.3 1509.81
    66.9 1510.65    80.2 1512.64    86.2 1513.28    98.1 1513.79   100.9 1514.13
   106.5  1515.2   108.7 1515.45   112.2 1515.65     115 1515.96     116 1516.14
   117.9 1516.77   126.3  1520.4     128 1520.96     134 1522.03   138.4 1522.51
#Mann= 3 ,-1,0
       0      .1       0    25.1    .045       0    59.2      .1       0
Bank Sta=26.4,59.4
XS Rating Curve= 0 ,0
Exp/Cntr(USF)=0,0
Exp/Cntr=0.3,0.1

Type RM Length L Ch R = 1 ,10477   ,97.4,91.8,85.6
XS GIS Cut Line= 2
2155132.25409538 627460.684345812155254.09652937627495.496469809
#Sta/Elev= 29
       0 1527.15     4.1 1524.37     8.2 1521.73    16.6 1517.13    20.7  1515.5
      23 1514.86    26.2 1513.84    33.2 1511.45    41.5 1507.31    45.7 1506.56
      54 1506.37    58.6 1506.39    62.3 1506.59    66.5 1507.05    70.6 1507.47
    74.8 1507.68      79 1507.59    83.1 1507.29    87.3 1507.39    91.4    1509
    95.6 1511.53    99.8 1513.46     104 1514.23   108.1 1514.72   112.2 1516.33
   116.4 1519.23   120.6 1521.25   124.7 1521.97   126.7 1522.01
#Mann= 3 ,-1,0
       0      .1       0    41.5    .045       0    66.5      .1       0
Bank Sta=41.5,66.5
XS Rating Curve= 0 ,0
Exp/Cntr(USF)=0,0
Exp/Cntr=0.3,0.1

Type RM Length L Ch R = 1 ,10385   ,78.6,79.4,77.2
XS GIS Cut Line= 4
2155102.12821884627565.1207178072155128.90677576627567.129109576
2155224.64011676627562.4428621152155262.13009645627552.400903269
#Sta/Elev= 30
       0 1532.37     2.1 1531.41     6.1 1528.61    10.8 1524.85    14.1 1522.41
    22.1  1516.8    34.1 1509.44    38.1 1507.31    42.1 1505.95    46.1 1505.45
    54.2 1505.47    70.2  1505.1    78.2  1505.2      83  1505.6    92.9 1506.01
    98.2 1505.95   102.2 1506.62   106.2 1507.93   110.2 1510.03   114.2 1511.87
   118.2 1512.39   126.4 1512.33   134.6 1512.62   139.7 1514.34   142.9 1515.61
   149.5 1517.02   151.2 1517.49   155.3 1519.05   158.5 1520.01   161.5 1520.55
#Mann= 3 ,-1,0
       0      .1       0    54.2    .045       0      83      .1       0
Bank Sta=54.2,83
XS Rating Curve= 0 ,0
Exp/Cntr(USF)=0,0
Exp/Cntr=0.3,0.1

Type RM Length L Ch R = 1 ,10305   ,82.5,75.8,74.8
XS GIS Cut Line= 4
 2155090.3415056627646.986856973 2155118.4424604627639.548368939
2155241.59076229627634.5893769162155318.45513864627609.794416803
#Sta/Elev= 30
       0 1523.31    14.3 1523.93    19.3 1523.33    22.6 1521.76    30.8 1513.69
    38.8 1505.34    42.8 1503.76    54.8 1502.73    58.8 1502.74    70.8 1503.25
    74.8 1504.25    78.8 1504.28    90.7 1501.83    98.9 1501.38   114.9 1501.84
   118.9  1503.2   126.9 1509.35   130.9 1510.36   142.9 1511.47   146.9 1511.45
   167.6 1509.84     176 1510.05   180.9 1511.47   192.9 1518.06   196.8 1519.21
   201.3  1519.8   205.5 1519.88   218.1 1519.09   226.5 1518.13   233.1 1518.38
#Mann= 3 ,-1,0
       0      .1       0    90.7    .045       0   114.9      .1       0
Bank Sta=90.7,114.9
XS Rating Curve= 0 ,0
Exp/Cntr(USF)=0,0
Exp/Cntr=0.3,0.1

Type RM Length L Ch R = 1 ,10230   ,76.1,81.3,83.4
XS GIS Cut Line= 3
2155132.98821536627722.8977388682155265.30106512627698.495778873
2155333.62655311627686.565931764
#Sta/Elev= 30
       0 1519.25     4.2 1518.75     7.3 1518.09    11.4 1516.02    16.8 1511.96
    19.5 1509.53    23.6 1505.23    27.6 1502.02    31.7 1500.13    35.8  1499.5
    39.8 1499.46      48 1499.72    56.1 1499.63    60.2 1499.78    64.3 1500.27
    72.4 1500.93    76.5 1501.53    88.7  1504.9    96.8 1506.88   100.9 1507.76
   104.9 1508.28   121.2 1508.94   129.3 1509.56   149.6 1508.49   162.4 1508.26
   165.9 1508.76     174 1512.07   178.1 1513.41   186.2 1514.55   203.9 1517.52
#Mann= 3 ,-1,0
       0      .1       0    31.7    .045       0    64.3      .1       0
Bank Sta=31.7,64.3
XS Rating Curve= 0 ,0
Exp/Cntr(USF)=0,0
Exp/Cntr=0.3,0.1

Type RM Length L Ch R = 1 ,10148   ,62.1,60.5,60.4
XS GIS Cut Line= 3
2155140.03767047627793.9345557442155244.15269979627793.392289966
2155328.20389533627808.033465964
#Sta/Elev= 30
       0 1516.04     8.1 1515.05    12.1 1513.35    16.1 1510.01    20.1 1505.72
    24.1 1501.83    28.1 1499.79      311498.956    36.1 1498.15    44.1 1498.06
    52.6 1498.14    56.6 1498.45    59.7 1499.08    67.7 1499.36    71.8 1499.78
    84.1 1502.07    92.1 1502.75   104.1  1505.4   108.2  1505.4   112.3 1504.82
   116.3 1503.93   120.4 1503.94   128.5 1505.53   148.8 1506.59   152.4 1507.26
   155.8 1508.55     161 1511.08     165 1513.56   173.1 1519.04   189.4 1529.35
#Mann= 3 ,-1,0
       0      .1       0      31    .045       0    59.7      .1       0
Bank Sta=31,59.7
XS Rating Curve= 0 ,0
Exp/Cntr(USF)=0,0
Exp/Cntr=0.3,0.1
